--- 72_ras.prj (project) ---

Proj Title=72
Current Plan=p01
Default Exp/Contr=0.3,0.1
English Units
Geom File=g01
Flow File=f01
Plan File=p01
Y Axis Title=Elevation
X Axis Title(PF)=Main Channel Distance
X Axis Title(XS)=Station
BEGIN DESCRIPTION:
RFD model 72 exported to HEC-RAS
END DESCRIPTION:

--- 72_ras.p01 (plan) ---

Plan Title=Plan 01
Program Version=4.10
Short Identifier=Plan 01
Geom File=g01
Flow File=f01
Subcritical Flow
Calc Critical at every XS
Secant Critical Depth

--- 72_ras.f01 (steady flow) ---

Flow Title=Flow 01
Program Version=5.01
Number of Profiles= 5
Profile Names=10yr,25yr,50yr,100yr,500yr
River Rch & RM=72,48,3022.565
  131.72   234.6  334.16  453.64  807.51
River Rch & RM=72,48,2702.075
  142.89  254.94  363.76  494.73  885.02
River Rch & RM=72,48,2579.157
   146.6  261.72  373.63  508.45  910.98
River Rch & RM=72,48,2479.741
  155.88  278.66  398.32  542.81  976.17
River Rch & RM=72,48,2331.605
  170.69  305.74  437.88  597.94 1081.26
River Rch & RM=72,48,2168.054
  172.54  309.13  442.82  604.84 1094.46
River Rch & RM=72,48,2078.701
  210.63  379.02  545.21  748.06 1370.12
River Rch & RM=72,48,1989.347
   224.7  404.92  583.26  801.44 1473.66
River Rch & RM=72,48, 1810.64
  228.98   412.8  594.85  817.71 1505.31
River Rch & RM=72,48,1737.093
  244.85  442.06  637.91  878.24 1623.32
River Rch & RM=72,48,1610.534
  260.69   471.3  681.01  938.91 1742.08
River Rch & RM=72,48,1427.325
  267.38  483.67  699.26  964.61 1792.54
River Rch & RM=72,48,1304.199
  269.81  488.17  705.89  973.97 1810.91
River Rch & RM=72,48,1113.455
   293.5     532  770.63 1065.33 1990.92
River Rch & RM=72,48,934.6901
  297.14  538.74   780.6  1079.4 2018.75
River Rch & RM=72,48,803.3347
  301.38   546.6  792.23 1095.84 2051.25
River Rch & RM=72,48,555.9908
  335.87   610.6  887.01 1229.95 2317.49
River Rch & RM=72,48,  346.76
  347.34  631.93  918.63 1274.77 2406.85
River Rch & RM=72,48,127.3899
  420.76  768.72 1121.99 1563.75 2987.05
Boundary for River Rch & Prof#=72,48,1
Up Type= 0
Dn Type= 2
Boundary for River Rch & Prof#=72,48,2
Up Type= 0
Dn Type= 2
Boundary for River Rch & Prof#=72,48,2
Up Type= 0
Dn Type= 2
Boundary for River Rch & Prof#=72,48,2
Up Type= 0
Dn Type= 2
Boundary for River Rch & Prof#=72,48,2
Up Type= 0
Dn Type= 2

--- 72_ras.g01 (geometry) ---

Geom Title=72
Program Version=4.10

River Reach=72,48
Reach XY= 30
1252154.90414336836742.7229910941252124.20215833836622.234148994
1252040.03551298836505.5675192481252005.03552279836488.900858521
1251964.20219964836426.4008781911251875.86889154 836403.06755434
1251797.53557849836311.4009170831251730.86893064836284.734260216
1251730.86892995836260.567600727 1251684.3877117836219.786417782
1251660.03561395836143.0676375481251545.69740942836021.204932943
 1251498.3689881835915.567709491 1251419.2023412835797.234413445
 1251295.8690415835708.0677767251251240.03571987835548.067825645
1251156.70241049835530.5678332451251090.03576195835483.067849264
1250948.36913568835440.5678659831250908.36914635835402.234545127
1250899.20247906835290.5679117441250862.53582132835228.067931265
1250862.53581962835168.9012820871250836.70249185835100.567969739
1250826.70249027834945.5680157991250796.70249763 834895.56803146
1250683.36919516834815.5680584461250590.86922157834788.068069249
1250424.20260361834779.7347432671250314.20263693834813.901403055

Type RM Length L Ch R = 1 ,3022.565,23.761100,23.761100,23.761100
XS GIS Cut Line= 6
1252260.54100623836721.8978689261252196.08620046836738.129330067
1252175.65645019836740.4379626971252146.55771702836740.563054911
1252127.49567169 836743.429693521252063.80947344836762.411041598
#Sta/Elev= 30
 9892.56398.56969911.285384.97649918.108380.73059928.333372.92929938.401366.3322
9945.113360.94879948.468358.50869951.824356.45769957.223 353.8389961.846351.9657
 9968.45350.48519971.751348.76499981.644341.38919984.924339.82739988.205339.0404
9991.486338.7179 9998.05337.156510007.89338.385610014.52339.834810024.47 342.525
10027.79343.610310031.18345.121410041.35352.414110044.74354.4975 10058.3361.9543
10061.72364.106110065.18366.680510079.02376.009610085.93380.104810094.49384.7381
#Mann= 3 , 0 , 0
 9892.56    0.12       0 9892.56    0.12       010094.49    0.12       0
#XS Ineff= 2 , 0
       09990.578                       0
Bank Sta=9892.56,10094.49
Exp/Cntr=0.3,0.1

Type RM Length L Ch R = 1 ,2998.804,24.988300,24.988300,24.988300
XS GIS Cut Line= 4
1252255.61623513836684.7531498731252160.59825466836715.886840618
1252158.72559632836716.5890875551252063.78214459836747.915285107
#Sta/Elev= 30
9897.007 392.5879900.417389.92069907.322383.86689914.227  378.71 9917.68375.7994
9924.585370.48499928.037368.12519938.394362.14279945.299357.85779955.657350.9295
9966.014 343.6579972.357339.47139976.372337.31769983.276333.97269993.634329.2848
9997.088327.925610000.57327.375710004.02327.754610014.39330.170410017.84331.2128
 10021.3332.553910024.75334.204310045.48345.101410052.39350.024410055.85352.1389
10062.76355.467410069.67358.170710080.03364.291410090.39 371.24410098.97 376.287
#Mann= 3 , 0 , 0
9897.007    0.12       09897.007    0.12       010098.97    0.12       0
#XS Ineff= 2 , 0
       09990.917                       0
Bank Sta=9897.007,10098.97
Exp/Cntr=0.3,0.1

Type RM Length L Ch R = 1 ,2973.816,24.703700,24.703700,24.703700
XS GIS Cut Line= 6
 1252240.7070042836655.0347993961252175.75734448836680.028322969
1252148.80736359836694.0058330611252147.14326303836695.115233506
1252125.07076838836707.1361206011252055.38907052836734.408639467
#Sta/Elev= 30
9899.048381.59299904.123377.62469918.184367.8753 9928.73360.31529932.245358.0243
9939.276353.89159942.792351.69769956.853341.79459963.884336.58799967.399334.2739
9971.031332.54789974.727 331.2059982.119328.92119993.206325.95779996.902325.1225
 10000.7324.573310004.46324.831110008.19325.710910011.93326.883610015.66328.3371
10026.83333.370610033.88336.310910051.49 342.74410058.54345.189910062.06346.6252
10065.58348.677610076.15356.3422 10083.1360.943510097.29 369.19710100.96371.6503
#Mann= 3 , 0 , 0
9899.048    0.12       09899.048    0.12       010100.96    0.12       0
#XS Ineff= 2 , 0
       09972.545                       0
Bank Sta=9899.048,10100.96
Exp/Cntr=0.3,0.1

Type RM Length L Ch R = 1 ,2949.112,24.703700,24.703700,24.703700
XS GIS Cut Line= 5
1252231.32619628836636.5003583791252137.93138096836672.197946869
 1252136.0744276836672.9407282761252098.19505819836687.342806364
1252043.59122662836710.894877084
#Sta/Elev= 30
9899.015375.90259908.092369.91289918.629361.57879922.141359.47639925.653357.1546
 9936.19349.21379939.703346.74049946.727 342.569 9950.24  339.889957.264333.8495
9964.289 327.4669967.801 325.294 9971.23323.42649974.826322.25019978.338321.5482
9981.851 321.052  9995.9319.847910002.94 319.53610006.45319.617110009.96320.2474
10016.98323.189810020.49324.327310034.52328.332110038.03329.651910041.55331.2267
10066.56343.406610069.37344.930710087.99356.777310095.14360.205810100.99 363.512
#Mann= 3 , 0 , 0
9899.015    0.12       09899.015    0.12       010100.99    0.12       0
#XS Ineff= 2 , 0
       09980.132                       0
Bank Sta=9899.015,10100.99
Exp/Cntr=0.3,0.1

Type RM Length L Ch R = 1 ,2924.408,24.703800,24.703800,24.703800
XS GIS Cut Line= 6
1252226.99341201836614.2686500861252162.60353146836641.009502976
1252145.90033589836645.9001693811252117.39371773 836651.44971951
1252101.95566474836656.4728726161252039.02827521836686.034961988
#Sta/Elev= 30
9899.031374.1478 9903.52371.57639907.072368.75879910.625366.27369914.177363.9752
 9931.94351.48189955.787335.01499956.807334.25479970.932322.10939977.769316.3992
9981.188315.20279991.324315.87099994.665 315.72710001.35 314.63110004.69314.2794
10008.03314.128910011.38314.1676 10015.2314.406110021.61315.422110025.06316.2042
10028.51317.121410031.98318.174610035.61319.6689 10045.1323.063310050.11324.9755
10060.53329.375310064.61331.323310075.48337.2552 10091.4345.481610100.96350.8601
#Mann= 3 , 0 , 0
9899.031    0.12       09899.031    0.12       010100.96    0.12       0
#XS Ineff= 2 , 0
       09986.669                       0
Bank Sta=9899.031,10100.96
Exp/Cntr=0.3,0.1

Type RM Length L Ch R = 1 ,2899.704,24.703700,24.703700,24.703700
XS GIS Cut Line= 4
1252214.55719267836577.6842901591252126.24659509836624.572812839
1252124.39723892836625.334312508   1252036.86562836673.597582225
#Sta/Elev= 30
9899.014368.0051 9900.77367.90879904.485366.44839911.508360.46479915.629357.6567
9919.343355.58839923.058353.1165  9925.5351.23939939.492339.44339945.346334.9418
9956.489 328.3249975.062316.30239982.492311.14729989.921305.40019993.635306.2266
 9997.35306.597710009.58306.867310016.37307.3741 10019.7307.784210023.45308.9402
10029.96312.027610034.69314.495410038.44316.184210042.18317.033510045.93317.4027
10049.68318.340510064.66325.4834 10075.9330.299410091.11338.393910100.96344.2687
#Mann= 3 , 0 , 0
9899.014    0.12       09899.014    0.12       010100.96    0.12       0
#XS Ineff= 2 , 0
       09989.563                       0
Bank Sta=9899.014,10100.96
Exp/Cntr=0.3,0.1

Type RM Length L Ch R = 1 ,2875.001,24.703700,24.703700,24.703700
XS GIS Cut Line= 6
1252192.12247484836552.9035372331252134.66675763836587.758922908
1252108.56754236836607.5785524541252106.97882673836608.793452713
1252079.97045553836628.5581220451252022.80203429836662.546696139
#Sta/Elev= 30
9899.027351.3006  9905.3348.65959909.137346.10239912.975343.12789916.812340.6197
9920.649338.48579928.324333.81459939.124327.79229951.348319.73039966.228310.7848
9970.107308.88869974.971307.14859979.091 305.8539986.382304.07789995.569302.3378
9999.691301.761110003.78301.485110008.24301.6737 10013.8302.820310024.91306.3304
10032.24308.877710036.19310.464710047.64315.705210059.09321.161710062.91323.1099
10078.17 333.45110081.99335.854510085.81337.783510093.44340.852310100.98344.1737
#Mann= 3 , 0 , 0
9899.027    0.12       09899.027    0.12       010100.98    0.12       0
#XS Ineff= 2 , 0
       09978.498                       0
Bank Sta=9899.027,10100.98
Exp/Cntr=0.3,0.1

Type RM Length L Ch R = 1 ,2850.297,24.703700,24.703700,24.703700
XS GIS Cut Line= 5
1252181.77745838836534.180545938 1252096.4896287 836586.37200145
1252094.84154488836587.5050591451252062.96789928836605.969052854
1252009.92669087836640.249761584
#Sta/Elev= 30
 9899.01342.31539908.556337.75029920.095  332.62 9924.44330.91639927.788329.2288
9939.327321.4706 9947.02316.59549958.559311.77719977.791301.96139981.637300.8665
9987.295297.9737 9989.33297.34849997.023296.284910008.52295.8412 10019.9296.4189
10023.69296.896510027.48299.236610032.37303.546310035.06305.486910038.88306.9854
10042.79306.2913 10046.7306.0937 10050.6307.440710056.96310.930110066.23316.9144
10070.14318.9628 10075.1321.176410081.14323.100110097.48328.920810100.99330.8368
#Mann= 3 , 0 , 0
 9899.01    0.12       0 9899.01    0.12       010100.99    0.12       0
#XS Ineff= 2 , 0
       0                10019.88       0
Bank Sta=9899.01,10100.99
Exp/Cntr=0.3,0.1

Type RM Length L Ch R = 1 ,2825.593,24.703700,24.703700,24.703700
XS GIS Cut Line= 6
1252169.27352418836513.189639656 1252106.3447544836553.713180912
1252084.07772262 836565.356620151252082.24358253836566.154072427
1252055.48288716836580.6093906791251998.53287296836620.507674598
#Sta/Elev= 30
9899.025 331.8799901.714 331.4929905.543330.59099909.446329.08029960.175 304.743
9971.881300.02989975.686298.0437 9983.09292.69519994.197 287.3069997.899287.0982
10001.54287.469810009.98288.883510016.45290.141510023.91291.832710027.64292.2014
10031.37291.934110035.37292.278110039.38 294.08310047.39298.037710051.39299.6398
 10055.4301.031510065.12304.009610067.42305.071310075.43309.378410079.43310.9879
10083.44311.808110087.45312.884110093.71314.988510095.46315.807710100.95319.0473
#Mann= 3 , 0 , 0
9899.025    0.12       09899.025    0.12       010100.95    0.12       0
#XS Ineff= 2 , 0
       0 9989.47        10020.23       0
Bank Sta=9899.025,10100.95
Exp/Cntr=0.3,0.1

Type RM Length L Ch R = 1 , 2800.89,24.703800,24.703800,24.703800
XS GIS Cut Line= 5
1252152.30310319836485.378399429 1252079.0802429836538.218537527
1252071.36979426836544.1065802441252069.79108986836545.334461521
1251990.45897973836606.192144659
#Sta/Elev= 30
9899.001315.51769905.061315.35299909.107314.55359917.199311.89389929.336308.5445
9941.474304.08399949.566300.69479957.658298.26819961.703296.22729965.749 293.699
9973.841289.23059981.933285.61919988.261283.35289993.704281.8396   10001281.0531
10009.87281.696110018.98283.292210027.25286.865310031.38288.460610035.52289.6832
10039.65290.556210042.21290.689910052.99 293.41910064.46295.2668 10068.6 296.435
10072.73298.341510076.87300.9226   10081304.863910085.14307.923910100.99310.5574
#Mann= 3 , 0 , 0
9899.001    0.12       09899.001    0.12       010100.99    0.12       0
#XS Ineff= 2 , 0
       09988.053                       0
Bank Sta=9899.001,10100.99
Exp/Cntr=0.3,0.1

Type RM Length L Ch R = 1 ,2776.186,24.703700,24.703700,24.703700
XS GIS Cut Line= 5
1252134.07020506836462.2722182651252055.99695413836524.751871532
1252054.43521655836526.0012616761252041.00487187 836536.72443974
1251979.29834232836591.948737712
#Sta/Elev= 30
9899.004 298.639 9911.36299.45639915.562299.55959919.816299.49849923.967299.1857
9928.169 298.3069935.568295.89179949.179291.03569953.381289.35749961.822285.5554
9967.073283.50119978.593279.86759982.826278.2019  9991.2273.77579993.327272.8332
9995.402272.08049999.604271.667510003.83271.8182 10012.2272.744310018.19273.8595
10033.92277.766510038.33278.481810047.13278.698810051.53279.453410055.94280.6452
10060.34282.512210069.15 286.86510086.76296.302510093.31 299.131   10101301.8303
#Mann= 3 , 0 , 0
9899.004    0.12       09899.004    0.12       0   10101    0.12       0
#XS Ineff= 2 , 0
       0                               0
Bank Sta=9899.004,10101
Exp/Cntr=0.3,0.1

Type RM Length L Ch R = 1 ,2751.482,24.703700,24.703700,24.703700
XS GIS Cut Line= 6
1252112.39844016836435.3044626051252062.76378297836481.210484806
1252040.99578319836505.1635803961252039.44355522836506.424765693
1252007.62140878836543.7040675611251971.52751302836579.687791053
#Sta/Elev= 30
9899.025280.5581 9904.99279.95079909.574279.93769914.406280.62079927.335283.3348
9933.734282.4704 9945.21 280.0839953.061277.75959963.086274.13859967.639271.9081
9977.396266.2607 9980.78264.73249987.152263.77659989.647  262.239992.031259.7727
 9994.08258.31159998.513256.4248 10001.5255.868210003.18256.157610006.55257.4676
10029.06268.453410036.87271.8302   10042271.704110050.01268.106610051.86268.1025
10055.33269.691610069.27278.305310084.29286.9954 10092.5 291.18910100.98294.5364
#Mann= 3 , 0 , 0
9899.025    0.12       09899.025    0.12       010100.98    0.12       0
#XS Ineff= 2 , 0
       0                               0
Bank Sta=9899.025,10100.98
Exp/Cntr=0.3,0.1

Type RM Length L Ch R = 1 ,2726.778,24.703700,24.703700,24.703700
XS GIS Cut Line= 6
1252083.81584063836418.7116694541252034.72098037 836467.94850663
1252024.47399682  836482.13440371252012.26008128836507.114034155
1252002.72269086836521.8134959671251955.94225003836573.201644009
#Sta/Elev= 30
9899.067265.15069904.815263.46879909.449263.39929914.082264.99029920.547268.3338
9923.348268.96789925.194269.03479932.614268.46739948.426266.26539951.147265.3297
9960.413260.37039967.012 257.732 9973.59254.51559977.637252.17819983.495 253.577
9986.097253.44979989.442 253.9599993.118249.32659996.795246.295510000.43246.7324
10004.06248.024410022.89256.765710030.71259.822210034.92260.787410046.29262.1133
 10051.4264.090110066.25 273.48510083.41 282.96110089.86285.986910100.97290.5741
#Mann= 3 , 0 , 0
9899.067    0.12       09899.067    0.12       010100.97    0.12       0
#XS Ineff= 2 , 0
       0                               0
Bank Sta=9899.067,10100.97
Exp/Cntr=0.3,0.1

Type RM Length L Ch R = 1 ,2702.075,24.703700,24.703700,24.703700
XS GIS Cut Line= 5
1252071.12658554836411.7311949231251998.70642204836480.687704054
1251997.24734767836482.0555863581251979.11452698836499.333405325
1251927.82965908836553.982326094
#Sta/Elev= 30
9899.002262.82919906.953 260.262 9910.27259.76739915.028260.31699916.014260.7417
9920.544261.64799925.074261.66499938.665 260.0569943.574260.18329947.725258.8607
9952.255256.39319957.848254.32419962.605251.12669972.121244.30569974.906242.4454
9976.879241.43829997.557233.805110000.68233.705410002.07233.952210005.44235.2426
10038.05249.569410043.83252.629610047.05255.024910048.63255.671210051.54255.6941
10056.04256.651910063.01260.271810074.04266.459310092.04274.792910100.99279.1923
#Mann= 3 , 0 , 0
9899.002    0.12       09899.002    0.12       010100.99    0.12       0
#XS Ineff= 2 , 0
       0                10015.47       0
Bank Sta=9899.002,10100.99
Exp/Cntr=0.3,0.1

Type RM Length L Ch R = 1 ,2677.371,24.703800,24.703800,24.703800
XS GIS Cut Line= 6
1252063.79136929836397.2578535831252012.49558262836444.208525256
1251970.85029785836467.9581686491251956.36241069836478.385800982
1251937.95297829 836496.493524561251911.69151829836527.537246305
#Sta/Elev= 30
9899.054264.17999905.812261.5493 9910.26260.18379923.603257.49429932.498255.2049
9951.436248.65299961.155246.95239963.631245.75639972.085240.05429991.517229.3911
9995.195228.20169998.874227.616110002.52227.393310006.22227.648510009.92228.3246
10016.62 230.15910021.43 231.99210025.47233.052810029.51232.279410034.71234.3822
10038.03235.424810044.07235.149110047.24235.313910048.75 235.74810051.84237.1339
 10058.1240.946310061.12 241.91710066.88243.111210071.17244.858510100.95 262.183
#Mann= 3 , 0 , 0
9899.054    0.12       09899.054    0.12       010100.95    0.12       0
#XS Ineff= 2 , 0
       0                 10014.4       0
Bank Sta=9899.054,10100.95
Exp/Cntr=0.3,0.1

Type RM Length L Ch R = 1 ,2652.667,24.703700,24.703700,24.703700
XS GIS Cut Line= 6
1252048.26772824836370.4381949721251998.72268493836420.143493315
1251963.45166245836445.5402162961251951.44980207836456.013917049
1251934.14494517836475.7090867681251906.20061875836512.357312423
#Sta/Elev= 30
9899.032267.27579907.341 264.6489916.635259.70859921.983256.3298 9925.93253.2848
9931.248248.14889935.224246.34529940.512246.09199944.519244.17489949.777240.0917
9953.814238.42969959.042237.62479963.674236.30289989.221225.42019995.171224.0179
    9999223.839110004.56224.501310007.25225.416110016.81230.255310018.04230.4462
10021.16229.821210025.52226.618510030.04225.032110036.83224.268310045.57224.9746
10060.31230.505810070.84233.914910074.96235.826110087.36 242.84710100.97252.0851
#Mann= 3 , 0 , 0
9899.032    0.12       09899.032    0.12       010100.97    0.12       0
#XS Ineff= 2 , 0
       0                10012.13       0
Bank Sta=9899.032,10100.97
Exp/Cntr=0.3,0.1

Type RM Length L Ch R = 1 ,2627.964,27.126100,27.126100,27.126100
XS GIS Cut Line= 6
1252013.52575773836339.0617759081251977.47400231836387.153980333
 1251956.7096256836421.1749322911251955.75192139836422.930723466
1251935.06480384836457.7703532261251901.61737669836506.936273039
#Sta/Elev= 30
9899.038275.76749905.593 270.9839909.363268.59789922.003261.98279929.865257.2709
9938.066252.71149949.351243.23719954.467240.18419959.143238.37179962.447236.6889
9966.291 233.816 9973.06227.50669977.821224.31599993.196218.2932 9998.25216.7221
10000.83216.357310004.64216.994910016.09220.999210019.91221.808810027.54222.5703
10043.17222.973810049.01223.459710050.79223.837210054.84226.212610058.72 228.062
10070.63230.873610078.56233.357710082.53 235.408 10086.5238.064510100.98248.8673
#Mann= 3 , 0 , 0
9899.038    0.12       09899.038    0.12       010100.98    0.12       0
#XS Ineff= 2 , 0
       0                10018.95       0
Bank Sta=9899.038,10100.98
Exp/Cntr=0.3,0.1

Type RM Length L Ch R = 1 ,2600.838,21.680100,21.680100,21.680100
XS GIS Cut Line= 6
1251950.16891864836362.8167793751251937.70110402836388.333179057
1251931.56350669836408.6193546651251925.98753995836444.691469625
1251918.75205392836465.0356813821251900.24557856836499.204472572
#Sta/Elev= 30
9944.131239.29989948.796 237.0919952.448235.54429956.099234.24169965.708231.0591
9970.705228.99039977.673225.87669984.528223.45859987.956221.89589993.725218.6905
9994.777 218.2019998.095  217.0410001.41217.178610004.73217.724210008.05216.7925
10011.35216.651810014.68216.8119   10018217.121710030.23218.6374 10041.8219.7897
10045.28220.249910048.76220.833310052.27222.2456   10056224.118910063.47226.9649
10070.93230.040510078.39233.811510082.12236.059610085.85238.907210090.68242.8401
#Mann= 3 , 0 , 0
9944.131    0.12       09944.131    0.12       010090.68    0.12       0
#XS Ineff= 2 , 0
       09990.241        10021.46       0
Bank Sta=9944.131,10090.68
Exp/Cntr=0.3,0.1

Type RM Length L Ch R = 1 ,2579.157,34.575600,34.575600,34.575600
XS GIS Cut Line= 6
1251945.64439297836337.151108325 1251915.9849332 836388.55258511
1251909.53476351836409.1607006641251905.35211831836445.412480533
1251899.86455089836465.8812138591251887.97941574836491.671979904
#Sta/Elev= 30
9914.795243.91319919.085241.15539922.984 238.9349926.883237.26729930.782  235.87
9934.681 234.174 9938.58232.18489950.263225.8895  9955.3223.89179968.517219.4135
9979.164215.5777 9990.36210.43919992.916208.98149995.831206.98169999.641204.6794
10002.95204.360410012.87208.195210019.46 210.37610029.37213.103310039.47215.4326
10042.87216.448510046.26  217.8510056.64222.665910063.86225.774210065.71226.7254
10067.48227.855910071.09230.838810073.55233.362310078.31238.856910081.92242.2229
#Mann= 3 , 0 , 0
9914.795    0.12       09914.795    0.12       010081.92    0.12       0
#XS Ineff= 2 , 0
       09990.221        10020.06       0
Bank Sta=9914.795,10081.92
Exp/Cntr=0.3,0.1

Type RM Length L Ch R = 1 ,2544.582,15.433100,15.433100,15.433100
XS GIS Cut Line= 6
1251942.34627301  836328.63155591251908.05807859836367.694055915
1251879.41224524836397.2079447951251867.69349524836422.381555915
1251849.03030077836465.7843336761251833.41723713836494.863358289
#Sta/Elev= 30
9900.029 244.2919911.804236.2774 9916.17233.53239920.535231.02939937.344221.9934
9951.093216.42579956.961 213.5669969.339206.79659978.483 201.2279980.514200.0815
9983.055199.07269985.224198.43219996.013 198.1689999.632198.208510003.25198.8837
10006.87199.905510010.49199.219410014.11199.090110017.73200.145610021.34201.7553
10027.12204.8409 10039.2212.027310042.77214.472510060.62227.4621 10064.2229.8336
10068.57232.140510078.86 236.47610082.73 238.54810089.81242.898910101.17250.1473
#Mann= 3 , 0 , 0
9900.029    0.12       09900.029    0.12       010101.17    0.12       0
#XS Ineff= 2 , 0
       09986.114        10017.56       0
Bank Sta=9900.029,10101.17
Exp/Cntr=0.3,0.1

Type RM Length L Ch R = 1 ,2529.149,24.703700,24.703700,24.703700
XS GIS Cut Line= 6
1251937.57196745836328.1975281241251876.80807859836381.148917034
1251871.02088258 836385.620841221251864.85521162836393.293216929
1251863.63231671 836394.875786961251801.54608083836473.265328184
#Sta/Elev= 30
9901.245241.00199905.388238.25059914.508231.75399920.369227.91059927.563223.7499
9931.915221.46349936.267219.57499940.619219.2446 9944.97218.24029950.332214.0456
9953.674211.67359970.307200.69199975.433197.66949980.295 195.4599985.546193.5438
9988.174192.90629994.742193.301410003.12192.2972 10007.3193.530810011.49 195.112
10015.67197.149710019.55 198.64510024.84200.329810028.23201.844610030.12202.9132
10045.97212.351110057.53219.512210070.08228.065410086.82 238.907   10101248.7147
#Mann= 3 , 0 , 0
9901.245    0.12       09901.245    0.12       0   10101    0.12       0
#XS Ineff= 2 , 0
       09986.288        10017.89       0
Bank Sta=9901.245,10101
Exp/Cntr=0.3,0.1

Type RM Length L Ch R = 1 ,2504.445,24.703700,24.703700,24.703700
XS GIS Cut Line= 6
1251918.57061481836305.4576459841251877.19180215836353.130528182
 1251861.1925802836367.0458957951251837.68931155836382.532515156
1251822.48581997836394.7925803281251774.56835028836445.642359615
#Sta/Elev= 30
9899.055233.1894 9902.36231.42689906.704229.95279910.347227.81619915.393224.0372
9919.737221.47489924.081   219.69928.426217.17079937.114209.99279940.378207.6207
9941.459207.19899945.803206.41729950.388203.60259954.492200.26419958.836197.3067
9962.181195.78699969.329191.80289982.373 185.7429989.169179.65719990.388179.1129
10002.15176.843110006.07177.772210023.39188.614410044.74201.0793 10063.4213.0144
10068.32216.986610073.24220.492210083.08 226.60310092.31231.887710100.97238.5844
#Mann= 3 , 0 , 0
9899.055    0.12       09899.055    0.12       010100.97    0.12       0
#XS Ineff= 2 , 0
       09984.226                       0
Bank Sta=9899.055,10100.97
Exp/Cntr=0.3,0.1

Type RM Length L Ch R = 1 ,2479.741,20.568900,20.568900,20.568900
XS GIS Cut Line= 6
1251909.12332233836286.6505496641251868.33026189836329.892837427
1251851.78041444836343.791107622 1251825.4128637 836361.14136881
1251810.01377669836373.5150335561251761.67343476836423.478332373
#Sta/Elev= 30
9899.045235.02949910.407225.48099915.188 222.2939919.969219.5863 9924.75215.1755
9929.532211.37039932.841209.27069941.862204.39359946.372201.48839950.882198.1306
9965.189188.28889975.393181.77929983.647176.82879987.591174.1737 9995.48167.4756
9998.288167.24579999.412167.363510007.21171.9235 10015.3177.2037 10019.5180.4452
10023.71182.876610036.25 188.158   10041 190.77610050.49197.477310064.38206.1645
10068.84208.786710078.84213.929510083.69217.024510093.39223.761110100.98228.5998
#Mann= 3 , 0 , 0
9899.045    0.12       09899.045    0.12       010100.98    0.12       0
#XS Ineff= 2 , 0
       09984.306                       0
Bank Sta=9899.045,10100.98
Exp/Cntr=0.3,0.1

Type RM Length L Ch R = 1 ,2459.172,28.838600,28.838600,28.838600
XS GIS Cut Line= 6
1251890.13957732836267.7051952781251829.47973812836330.175551462
1251821.43110963836340.2552896511251820.31216392836341.912986999
 1251812.4182275836352.1182943611251753.43071791 836416.16594972
#Sta/Elev= 30
9900.448228.78849906.245 224.2299915.391216.38659922.066211.4102 9929.11205.4847
9947.402193.02179950.323190.77559959.742182.60379964.452 178.8349965.695178.0506
9970.268175.81389978.581173.36969988.055171.42119993.313170.65969998.571170.3463
10001.03170.370610005.11170.861810009.26 172.15110015.32175.833310024.53180.5124
10031.11184.456410040.03 189.34210057.87200.832810066.79204.7544 10077.8210.0924
10080.17211.492510084.63214.627210093.55221.224410097.17223.5654 10102.4226.1169
#Mann= 3 , 0 , 0
9900.448    0.12       09900.448    0.12       0 10102.4    0.12       0
#XS Ineff= 2 , 0
       09989.251                       0
Bank Sta=9900.448,10102.4
Exp/Cntr=0.3,0.1

Type RM Length L Ch R = 1 ,2430.334,26.474000,26.474000,26.474000
XS GIS Cut Line= 6
1251873.71703323 836247.678515651251819.50267691836305.456396741
1251803.40930923836318.5189030731251801.73785857836319.617198444
1251788.65442808836330.6895613641251736.53894969836395.024519551
#Sta/Elev= 30
9899.042 224.5099916.229211.5949 9923.21205.48999925.819203.37089941.206193.4725
9945.705190.02979954.703181.94319959.202178.57129968.971  171.759973.766167.5471
9982.235167.87879987.441167.51429991.203166.40729992.647 164.5789995.429162.3174
9999.608161.3239   10001161.297710003.77161.681210008.07162.797810012.37164.5168
10018.14167.896710039.55181.464310042.42182.926310047.63186.798110058.05193.1294
10063.26195.661910073.69199.548310081.77202.833510090.21206.995410100.93213.0903
#Mann= 3 , 0 , 0
9899.042    0.12       09899.042    0.12       010100.93    0.12       0
#XS Ineff= 2 , 0
       0 9990.07                       0
Bank Sta=9899.042,10100.93
Exp/Cntr=0.3,0.1

Type RM Length L Ch R = 1 , 2403.86,24.687100,24.687100,24.687100
XS GIS Cut Line= 6
1251840.60559652836224.1226116821251799.38743809836272.179676583
1251789.16839076836288.8220758361251764.53310625836338.579606084
1251747.23175456836363.6239502461251726.44452257836389.339025435
#Sta/Elev= 30
9900.358 211.7039907.609206.09649917.326199.20059922.185196.08629925.052194.3613
9931.903191.12549946.583181.78239954.946176.98929958.044174.66829967.191169.0898
9971.041166.96469975.806163.40259978.741160.36399982.076156.07519986.265153.2785
9989.902152.084710004.53150.570710008.15150.388910011.82152.121310015.49156.2723
10026.51167.928110030.19171.735410033.86174.934210049.39184.361810057.37 188.912
10065.34192.664110077.78 197.31610085.03200.552210090.25203.264410102.27210.4177
#Mann= 3 , 0 , 0
9900.358    0.12       09900.358    0.12       010102.27    0.12       0
#XS Ineff= 2 , 0
       09988.536                       0
Bank Sta=9900.358,10102.27
Exp/Cntr=0.3,0.1

Type RM Length L Ch R = 1 ,2379.173,22.950000,22.950000,22.950000
XS GIS Cut Line= 6
1251813.88540361836223.1478104351251766.64246134836277.777423846
1251760.00157836836290.9310275531251745.28101768836336.470771335
1251728.42435338836361.9167916681251705.26360119836389.864347987
#Sta/Elev= 30
9904.442194.07479908.244191.41889912.724188.58859921.683182.28319925.394180.1553
 9939.85172.47189944.669169.65459960.443159.78699965.077157.19879969.236155.1405
9973.395153.44759981.134151.6428 9984.81150.17519998.884147.386410002.27147.2303
10005.66149.112710009.04152.929510012.42156.4779 10015.8159.879510020.42164.1095
10029.85171.417610033.42173.693210040.69177.619910053.96185.591410065.84191.8019
10076.68196.181710085.13200.3855 10089.4202.311410097.25206.4231 10106.3210.3529
#Mann= 3 , 0 , 0
9904.442    0.12       09904.442    0.12       0 10106.3    0.12       0
#XS Ineff= 2 , 0
       09985.577                       0
Bank Sta=9904.442,10106.3
Exp/Cntr=0.3,0.1

Type RM Length L Ch R = 1 ,2356.223,24.617800,24.617800,24.617800
XS GIS Cut Line= 4
1251808.42775078836218.708575043 1251737.9719761 836289.56693705
1251736.66211507836291.0783152561251666.98780039836362.783465925
#Sta/Elev= 30
9899.075 190.6579904.636186.69299925.526175.16699939.485166.57649941.649165.1453
9948.791159.45179953.444156.30439969.409147.27149978.662141.46049981.362140.7082
9983.289140.98439986.016143.51589990.669146.18339992.542146.83659997.169144.6625
    9999143.2711   10001142.499110001.66142.429110004.81143.216310006.23  143.89
10015.38149.067210019.95152.044410023.65154.853810028.35160.748310042.48166.0388
10047.19168.1767 10056.6173.337610079.42184.169210089.56190.575410100.98  199.05
#Mann= 3 , 0 , 0
9899.075    0.12       09899.075    0.12       010100.98    0.12       0
#XS Ineff= 2 , 0
       09975.998        10009.95       0
Bank Sta=9899.075,10100.98
Exp/Cntr=0.3,0.1

Type RM Length L Ch R = 1 ,2331.605,24.789700,24.789700,24.789700
XS GIS Cut Line= 4
1251802.15530077836214.4822503631251750.81443909836255.974176913
1251727.96593156836271.4872739611251666.73863411836335.576000348
#Sta/Elev= 30
9911.127187.56179918.604181.98029922.823179.19549931.259175.08059935.477172.3748
9945.002 164.7429952.351159.59599956.569 156.923  9971.1148.6414 9985.56140.0391
9989.526 137.9149993.492136.06689997.457135.657210004.76138.154510009.81 140.719
10015.01144.052410018.89145.040710024.51145.445710029.26146.0959 10032.5146.9881
10034.01147.625410037.04149.482210038.76151.083410043.51150.688210048.26152.6343
10059.73161.246210064.26163.849910077.87 170.54210086.25175.998310093.39181.1718
#Mann= 3 , 0 , 0
9911.127    0.12       09911.127    0.12       010093.39    0.12       0
#XS Ineff= 2 , 0
       0                10015.27       0
Bank Sta=9911.127,10093.39
Exp/Cntr=0.3,0.1

Type RM Length L Ch R = 1 ,2306.815,24.703700,24.703700,24.703700
XS GIS Cut Line= 5
1251794.80868808836181.2127799451251720.30451101836247.883829141
1251718.84811107836249.2545585841251710.18809953 836257.17626324
1251640.01115325836310.685481303
#Sta/Elev= 30
 9899.02189.07139910.174184.99189911.963183.83449918.979178.11449932.187170.8268
9936.562168.10539946.402160.57879951.322157.04439958.603152.01049966.082147.1225
9975.922141.51189985.762135.38459995.601129.89739998.227128.920810000.48128.5778
10002.69128.616710015.32131.157310020.73 132.06710024.05132.027410028.17134.3892
10031.55138.2986 10032.3139.488810036.42139.779610040.55137.832410042.37138.2797
10044.67139.407510069.43158.248410081.81167.188110085.66169.663910100.99177.4806
#Mann= 3 , 0 , 0
 9899.02    0.12       0 9899.02    0.12       010100.99    0.12       0
#XS Ineff= 2 , 0
       0                10019.13       0
Bank Sta=9899.02,10100.99
Exp/Cntr=0.3,0.1

Type RM Length L Ch R = 1 ,2282.111,24.703700,24.703700,24.703700
XS GIS Cut Line= 6
1251777.16223361836165.6483450171251720.75233826836210.881323621
1251702.01913347836231.2175888341251700.72220056836232.740075298
1251679.94031984836254.6166933591251624.54973044836297.036590467
#Sta/Elev= 30
9899.045180.23759912.311171.64329929.133 161.6239933.338158.99239950.159 148.103
9954.365145.30769962.776139.47549966.981136.9236 9971.35133.88159976.004 130.894
9987.354  125.189991.814122.66929995.373121.49729996.275121.381810000.27121.8136
10005.19122.896510009.71124.124610028.89129.803110031.17130.388110037.46131.4505
10037.96 131.63610041.59133.653510043.35135.153710054.14143.561510070.33155.9013
10074.65159.076710087.05167.225410095.31172.965110097.31 174.16910100.94175.7198
#Mann= 3 , 0 , 0
9899.045    0.12       09899.045    0.12       010100.94    0.12       0
#XS Ineff= 2 , 0
       0                10021.56       0
Bank Sta=9899.045,10100.94
Exp/Cntr=0.3,0.1

Type RM Length L Ch R = 1 ,2257.408,89.353500,89.353500,89.353500
XS GIS Cut Line= 2
1251761.61457449836162.3848111331251592.34374118836278.704255566
#Sta/Elev= 30
 9904.78170.17299918.377161.58629938.281 148.3239946.243143.32639950.223140.4707
9962.166131.33729964.849129.66739966.147128.94279970.127127.12459978.089123.7913
9982.228121.63549994.012114.89839997.993113.458510001.97112.977510005.95113.9013
10009.94115.867510016.99118.766310021.88121.300310028.57125.227410033.82128.5927
 10037.8131.364310045.95137.320610051.74139.795510065.67145.026810073.63148.6219
10077.61151.567210089.55162.974110093.53166.507110101.49172.299310110.16178.1133
#Mann= 3 , 0 , 0
 9904.78    0.12       0 9904.78    0.12       010110.16    0.12       0
#XS Ineff= 2 , 0
       0                10019.62       0
Bank Sta=9904.78,10110.16
Exp/Cntr=0.3,0.1

Type RM Length L Ch R = 1 ,2168.054,89.353600,89.353600,89.353600
XS GIS Cut Line= 6
1251773.15103369836044.4377531171251669.94595699836118.644980905
1251652.30121689836133.183703205 1251650.8293549836134.537816309
1251637.49066322836145.3545999151251526.29225717836217.936047116
#Sta/Elev= 30
9849.023178.79319868.953170.64579872.994168.71479877.035166.09639885.117162.3113
9890.159159.50019909.362147.76389917.444143.69119925.525139.01519933.607134.9757
9941.689130.25849953.812123.92199969.975114.60689982.408108.35559986.659105.2915
 9990.91103.63489995.161103.207810003.74103.084310021.54 103.85310032.21104.8083
10036.13105.894110040.05 107.684 10051.8114.252110067.47124.147210075.56128.3297
10093.56139.311710102.73144.244310114.49 149.92410126.24157.170710150.96171.6578
#Mann= 3 , 0 , 0
9849.023    0.12       09849.023    0.12       010150.96    0.12       0
#XS Ineff= 2 , 0
       0                10023.57       0
Bank Sta=9849.023,10150.96
Exp/Cntr=0.3,0.1

Type RM Length L Ch R = 1 ,2078.701,89.353500,89.353500,89.353500
XS GIS Cut Line= 6
1251716.46914392835973.383373433 1251616.0904879836051.376405858
1251595.13460204836064.7260375131251577.73496146836076.070898995
1251527.04061535   836117.6302711251476.58407798836156.422496656
#Sta/Elev= 30
 9849.03134.63699851.753133.81919855.907133.49699860.062 132.4479868.372128.4361
9880.836124.41099891.685125.00679897.455124.03439907.727120.27979918.229115.7757
9926.539113.33239951.467103.00759955.622101.71499963.931100.17459966.54799.19986
9992.00888.45392    9999 87.946410007.8288.4383610021.7790.2852710036.0692.76222
10044.5595.5916610048.7995.0411210071.85108.799310091.12121.208810092.76122.5475
10095.26125.3274 10099.4128.448110114.29136.542610125.06143.965510150.97157.1377
#Mann= 3 , 0 , 0
 9849.03    0.12       0 9849.03    0.12       010150.97    0.12       0
#XS Ineff= 2 , 0
       0                10029.69       0
Bank Sta=9849.03,10150.97
Exp/Cntr=0.3,0.1

Type RM Length L Ch R = 1 ,1989.347,89.353500,89.353500,89.353500
XS GIS Cut Line= 6
1251659.61638062835919.6319261161251566.32801275835983.671586421
1251534.62488986836002.4010346661251532.82184377836003.266496857
1251490.71532987836027.7858634441251406.90240399836084.581770446
#Sta/Elev= 30
9849.024136.89649851.114 135.6599856.911131.02559858.283130.11269866.242125.7891
 9882.16115.33879890.119110.39369906.036101.32399917.97595.368499925.934 92.0456
9932.27290.304799945.83187.34456 9953.7984.784429961.749 82.6196 9977.0179.56878
9986.95577.039429996.06375.9295310007.3875.4707510018.7775.7783910026.36 76.4497
10045.7881.4973910049.1482.4307910052.0483.53721   1006188.5182610076.8696.51367
10088.74 102.85810112.52116.715910120.45121.092610140.27131.046810150.97136.7628
#Mann= 3 , 0 , 0
9849.024    0.12       09849.024    0.12       010150.97    0.12       0
#XS Ineff= 2 , 0
       0                10031.67       0
Bank Sta=9849.024,10150.97
Exp/Cntr=0.3,0.1

Type RM Length L Ch R = 1 ,1899.994,89.353600,89.353600,89.353600
XS GIS Cut Line= 6
1251629.87104846835842.4701796561251553.27777215835891.031186422
1251501.46124388835919.8292650361251499.64887762 835920.67503602
1251430.79859812 835959.331810081251371.20856819835997.953287395
#Sta/Elev= 30
9849.028131.92539865.578123.84969873.348 119.0919878.926115.40299888.886110.3651
 9900.54 105.8399921.81696.981069931.61791.936859946.90584.946389954.41281.14982
9961.91977.856089980.68667.972389988.19364.250279991.94762.63639  9995.761.74983
10003.1461.00087 10006.960.9497710010.6661.33336   1003765.4321210041.4965.61819
10052.0563.9499810055.82 63.7001 10067.164.8664510070.8765.6915610074.63 67.0386
10086.1572.3914510101.7977.7561210113.5282.9007210133.0694.1309410150.97103.2828
#Mann= 3 , 0 , 0
9849.028    0.12       09849.028    0.12       010150.97    0.12       0
#XS Ineff= 2 , 0
       0                               0
Bank Sta=9849.028,10150.97
Exp/Cntr=0.3,0.1

Type RM Length L Ch R = 1 , 1810.64,73.546600,73.546600,73.546600
XS GIS Cut Line= 6
1251576.01702541835759.4786955111251506.64176661835808.779165812
1251452.73831696835844.9022651571251451.07421641  835846.0116656
1251406.52251972835876.4160504141251330.43962139835935.035600691
#Sta/Elev= 30
9849.003132.90049860.456  125.969868.506121.78979880.581114.5776 9888.63110.1864
 9904.73100.91159916.805  93.1719936.87681.003139940.82678.901479948.72475.39405
9956.62372.361469988.02859.397439993.92156.122189996.11755.164719999.81854.80865
10011.4856.1861910031.8358.0621710047.7257.90259 10057.858.5793310068.5558.91319
 10079.358.8649610090.0659.1157210095.4359.7089810100.8161.5161910109.5464.84676
10117.8267.4624110121.9669.0097110133.0675.5133310142.6781.6111210150.9885.73898
#Mann= 3 , 0 , 0
9849.003    0.12       09849.003    0.12       010150.98    0.12       0
#XS Ineff= 2 , 0
       0                10063.74       0
Bank Sta=9849.003,10150.98
Exp/Cntr=0.3,0.1

Type RM Length L Ch R = 1 ,1737.093,126.559100,126.559100,126.559100
XS GIS Cut Line= 2
1251452.40723741 835736.665662841251307.00793186835901.596218407
#Sta/Elev= 30
9934.62673.114069940.42770.805089945.38869.123279957.05866.057879965.80663.43572
 9970.1861.955969975.15659.899819987.674 54.14699990.03953.186819992.04852.53038
    999551.778619999.96251.29683 10000.851.3048610013.9253.1078510022.6654.71773
10027.0455.1696310040.1655.0419110054.5453.6765110062.0352.78142 10066.452.58849
10079.3452.8218310094.2254.2337810097.0254.3904610105.76 54.449610114.5155.16401
10119.03 55.990510133.9162.4260310138.8864.7789910145.1368.22613 10154.573.07143
#Mann= 3 , 0 , 0
9934.626    0.12       09934.626    0.12       0 10154.5    0.12       0
#XS Ineff= 2 , 0
       0                10089.49       0
Bank Sta=9934.626,10154.5
Exp/Cntr=0.3,0.1

Type RM Length L Ch R = 1 ,1610.534,183.209200,183.209200,183.209200
XS GIS Cut Line= 2
1251385.13293186835621.6483017651251209.35168186835828.896565631
#Sta/Elev= 30
 9875.0480.575819878.40778.614179884.44574.495979893.04969.175389897.35166.98615
9905.95563.017219910.25761.214719918.86158.467999927.46555.416869931.76754.09611
9936.06953.035169939.27352.568659954.48951.07346 9979.8547.488629984.92246.52454
9989.99445.131989996.29742.1944810000.1442.02973 10004.9 42.7921 10009.2 44.2099
 10013.545.1425310020.4346.50465 10025.547.1095210047.9246.4386510069.4347.14067
10086.3646.6686410095.2446.8418210099.5448.1089510121.8757.9065710146.7969.33623
#Mann= 3 , 0 , 0
 9875.04    0.12       0 9875.04    0.12       010146.79    0.12       0
#XS Ineff= 2 , 0
       0                 10102.9       0
Bank Sta=9875.04,10146.79
Exp/Cntr=0.3,0.1

Type RM Length L Ch R = 1 ,1427.325,123.126400,123.126400,123.126400
XS GIS Cut Line= 2
1251270.19084062835506.8479163751251095.41939019 835736.66566285
#Sta/Elev= 30
9948.84252.623799952.25451.082169957.67448.959919961.93946.848649970.18344.25425
9973.93443.199329984.77441.29797 9986.6740.541169994.91338.7999110003.1636.49588
10007.2836.56857 10011.437.3889310015.5237.8520810023.7738.0246610033.5538.69234
10052.6238.9613910060.8638.1875510085.5937.8296910102.08 37.121910122.6938.22777
10139.1738.7761910152.7939.1688510169.05 39.172910184.5140.1289410192.7639.76823
10196.8840.3810510209.2443.7855410212.4145.1655210229.8555.4485910237.5760.24254
#Mann= 3 , 0 , 0
9948.842    0.12       09948.842    0.12       010237.57    0.12       0
#XS Ineff= 2 , 0
       0                10123.14       0
Bank Sta=9948.842,10237.57
Exp/Cntr=0.3,0.1

Type RM Length L Ch R = 1 ,1304.199,190.744100,190.744100,190.744100
XS GIS Cut Line= 2
1251207.18154296835400.2941350641251024.88987628835648.775037855
#Sta/Elev= 30
9863.94952.724259871.84949.668329895.09841.478119903.23639.655139907.30538.50869
9910.67437.298929919.51234.591519923.58133.844699935.78932.565399947.99632.52142
9966.13931.270419971.68631.279069977.23231.553639984.61731.506919988.325 30.7733
9992.75529.615029996.82428.883219999.41828.9060310009.03 29.8566 10021.630.65127
10033.4530.3082410043.7930.8021710054.8831.5921610077.0732.4142310094.4833.59611
10110.7635.1914110115.8935.8293110126.9937.5901910139.2439.9096710172.1348.54027
#Mann= 3 , 0 , 0
9863.949    0.12       09863.949    0.12       010172.13    0.12       0
#XS Ineff= 2 , 0
       09941.914        10044.09       0
Bank Sta=9863.949,10172.13
Exp/Cntr=0.3,0.1

Type RM Length L Ch R = 1 ,1113.455,178.764600,178.764600,178.764600
XS GIS Cut Line= 2
1251111.69543183835261.4052461831250878.40550131835526.162190631
#Sta/Elev= 30
9759.02756.658779780.84143.528699785.428 40.98439798.33234.699479807.07730.92664
9815.82327.539619820.196 26.38239828.94124.791849835.05424.132239849.94223.83431
9863.92322.975449869.79222.814549907.65123.896389916.39723.973689929.34323.74634
9973.243 24.07799978.96923.758949986.36123.082989990.73422.406899999.47920.55756
10003.7821.0939710016.9723.4667510021.3423.9303810051.9525.0737510063.3325.83568
 10068.326.3884610086.9330.5217110091.31 31.701410104.4335.99317 10111.938.79002
#Mann= 3 , 0 , 0
9759.027    0.12       09759.027    0.12       0 10111.9    0.12       0
#XS Ineff= 2 , 0
       09894.582        10051.36       0
Bank Sta=9759.027,10111.9
Exp/Cntr=0.3,0.1

Type RM Length L Ch R = 1 ,934.6901,131.355400,131.355400,131.355400
XS GIS Cut Line= 2
 1251056.3568902835193.0458711831250702.62425128835395.953857288
#Sta/Elev= 30
 9816.65 55.22959825.92750.065429841.05638.689249844.83836.481269867.53226.11736
9871.31424.722399878.87922.641349886.44321.016689916.70216.081169943.17816.69194
9950.74216.371269962.08915.329799969.65415.38874    998114.967769996.12913.57523
9999.91213.66977 10013.3 15.808810026.3915.9256110037.7316.4553810052.8616.03269
10112.2115.5460110139.8614.7393110158.7717.8644910170.1120.0993210184.7423.86535
10196.5926.4396610200.3728.0530310207.9431.8952710219.2835.4036210224.4537.46793
#Mann= 3 , 0 , 0
 9816.65    0.12       0 9816.65    0.12       010224.45    0.12       0
#XS Ineff= 2 , 0
       09943.215                       0
Bank Sta=9816.65,10224.45
Exp/Cntr=0.3,0.1

Type RM Length L Ch R = 1 ,803.3347,247.343900,247.343900,247.343900
XS GIS Cut Line= 2
1251061.78223741835056.3271211981250598.45758465 835309.14830175
#Sta/Elev= 30
9770.98654.618749781.23651.043479793.80947.552329812.49639.797999831.18432.76694
9849.87126.480619870.27820.373699883.50918.254269890.98416.575429902.19615.00176
9918.22412.126979938.77211.167139976.94611.654069984.42110.774049999.3717.716221
10003.118.50862210006.8510.0809310010.58 10.932210047.96 11.537710062.0610.77412
10077.869.18833710089.078.79407710100.289.938012 10141.48.36132310182.518.844909
10193.72 9.41557 10219.613.7196410234.83 17.080510264.7324.65564 10298.835.22762
#Mann= 3 , 0 , 0
9770.986    0.12       09770.986    0.12       0 10298.8    0.12       0
#XS Ineff= 2 , 0
       09961.159                       0
Bank Sta=9770.986,10298.8
Exp/Cntr=0.3,0.1

Type RM Length L Ch R = 1 ,555.9908,209.230800,209.230800,209.230800
XS GIS Cut Line= 2
1250954.95727247834766.8033740821250524.40171692835270.275596291
#Sta/Elev= 30
9788.95743.160139796.483 43.1938  9800.842.370929816.95436.285219822.38533.94801
9832.09828.815569842.19424.718629861.23719.082149872.48216.728079895.7729.857683
9917.9147.5120989938.9416.5279749960.5266.1197159988.5863.08711110020.963.790515
10059.264.02361110089.553.47007710129.934.134415 10159.13.45737510189.324.081386
10205.653.84945810240.994.70363510271.27 4.2915110316.71 5.7915510340.417.490173
10372.2310.5999410383.5813.6737210396.5315.7722810418.1222.9728710451.4234.89016
#Mann= 3 , 0 , 0
9788.957    0.12       09788.957    0.12       010451.42    0.12       0
#XS Ineff= 2 , 0
       0                10318.54       0
Bank Sta=9788.957,10451.42
Exp/Cntr=0.3,0.1

Type RM Length L Ch R = 1 ,  346.76,219.370100,219.370100,219.370100
XS GIS Cut Line= 2
1250757.04060584834534.164485186 1250472.3183836835277.220040724
#Sta/Elev= 30
9712.88635.030439722.203 33.22489736.25728.814519764.36523.110879774.90520.08724
9785.44519.175189799.49916.618969852.201 10.38619918.9564.1081969950.5771.691504
 9980.821.9022449996.2520.69684110041.932.98282710126.251.08146310143.821.844573
10189.491.67677810203.54 0.9683410214.091.445873 10270.31.74319610291.381.356044
10340.572.31935910361.651.86165910393.276.06717910410.847.25076910424.8910.12292
10435.4313.9203210445.9716.43234   1045318.9145610484.6231.9633110508.6242.82162
#Mann= 3 , 0 , 0
9712.886    0.12       09712.886    0.12       010508.62    0.12       0
#XS Ineff= 2 , 0
       0                10289.48       0
Bank Sta=9712.886,10508.62
Exp/Cntr=0.3,0.1

Type RM Length L Ch R = 1 ,127.3899,93.722900,93.722900,93.722900
XS GIS Cut Line= 2
1250458.41128832834617.3080239591250372.78608784835274.609565169
#Sta/Elev= 30
9836.951 42.06779847.90236.046089867.75325.898839877.67921.614759890.913 15.4262
9900.83911.291539907.4568.7440799930.6161.3192779933.9240.4779059937.2330.360892
10344.180.360892 10350.80.47225610357.420.88025810360.730.88459210370.651.643366
10383.89 2.24742 10390.53.20761210403.746.33498510410.367.62948110413.668.082579
 10426.99.29427410430.2110.1105310446.7518.9499810450.0620.5144510453.3721.72843
10456.6822.5469710469.9125.0898710476.5326.7338910496.3834.4216710499.8136.21163
#Mann= 3 , 0 , 0
9836.951    0.12       09836.951    0.12       010499.81    0.12       0
#XS Ineff= 2 , 0
       0                10114.72       0
Bank Sta=9836.951,10499.81
Exp/Cntr=0.3,0.1

Type RM Length L Ch R = 1 ,  33.667,0.000000,0.000000,0.000000
XS GIS Cut Line= 6
1250317.64069059834629.2259589731250329.94335085834728.983147323
1250363.69790787834878.4004361181250330.71179676834999.928213909
1250191.82290787835190.9004361181250216.12846339835302.011547223
#Sta/Elev= 30
9822.12735.243389837.54331.268549850.72728.795229860.615 26.35789883.74117.44052
9903.6618.2723769906.9817.1033079913.6215.7181729916.9415.383079  9930.35.458712
9947.0745.9405979980.7583.854171 10004.51.112212 10028.23.42398810041.745.509981
10061.867.158228 10071.86.55566910101.957.52133710118.757.09321110159.398.469353
10176.748.02633310204.838.962656 10221.5 8.1994210268.819.22584310312.059.496813
10365.868.60280510460.159.71680710473.5814.0319510507.1627.8785110552.1339.87082
#Mann= 3 , 0 , 0
9822.127    0.12       09822.127    0.12       010552.13    0.12       0
#XS Ineff= 2 , 0
       0                10050.33       0
Bank Sta=9822.127,10552.13
Exp/Cntr=0.3,0.1
